--- GLADERN.prj (project) ---

Proj Title=GLADERN
Current Plan=p01
Default Exp/Contr=0,0
English Units
Geom File=g01
Flow File=f01
Plan File=p01
Background Map Layer=Inundation Boundary (01pct Value_0)
Background Map Layer=Inundation Boundary (01pct Value_0)
Background Map Layer=Inundation Boundary (01pct Value_0)
BEGIN DESCRIPTION:
----------MODEL BY WOOD PLC 2021----------
Stream Name: Glade Run
Flood Zone: Enhanced Approximate
Pocahontas County, WV
HEC-RAS Version: RAS 6.1
Vertical Datum: NAVD88
Projection: NAD 1983 StatePlane West Virginia S FIPS 4702 (US Feet)
Terrain: 1-meter LIDAR (FEMA Region III 3DEP collected 2016-2018)
Land Use: 2019 NLCD
Hydrologic Method:
WV SIR2010-5033 regression equations
END DESCRIPTION:
DSS File=dss
DSS Export Rating Curves= 0
DSS Export Rating Curve Sorted= 0
DSS Export Volume Flow Curves= 0
DXF OffsetX= 0
DXF OffsetY= 0
DXF ScaleX= 0
DXF ScaleY= 0

--- GLADERN.p01 (plan) ---

Plan Title=Floodplain
Program Version=6.10
Short Identifier=Floodplain
Geom File=g01
Flow File=f01
Subcritical Flow
K Sum by GR= 0
Std Step Tol= 0.01
Critical Tol= 0.01
Num of Std Step Trials= 20
Max Error Tol= 0.3
Flow Tol Ratio= 0.001
Split Flow NTrial= 30
Split Flow Tol= 0.02
Split Flow Ratio= 0.02
Log Output Level= 0
Friction Slope Method= 1
Unsteady Friction Slope Method= 2
Unsteady Bridges Friction Slope Method= 1
Parabolic Critical Depth
Global Vel Dist= 0 , 0 , 0
Global Log Level= 0
CheckData=True
Encroach Param=-1 ,0,0, 0
Computation Interval=0.1SEC
Output Interval=1SEC
Instantaneous Interval=Max Profile
Mapping Interval=1HOUR
Computation Time Step Use Courant=        0
Computation Time Step Use Time Series=    0
Computation Time Step Count To Double=0
Computation Time Step Max Doubling=0
Computation Time Step Max Halving=0
Computation Time Step Residence Courant=0
Run HTab= 0
Run UNet= 0
Run Sediment= 0
Run PostProcess= 0
Run WQNet= 0
Run RASMapper=-1
UNET Theta= 0
UNET Theta Warmup= 0
UNET ZTol= 0
UNET ZSATol= 0
UNET MxIter= 0
UNET Max Iter WO Improvement= 0
UNET MaxInSteps= 0
UNET DtIC= 0
UNET DtMin= 0
UNET MaxCRTS= 0
UNET WFStab= 0
UNET SFStab= 0
UNET WFX= 1
UNET SFX= 1
UNET Gravity=32.174
UNET 1D Methodology=Finite Difference
UNET DSS MLevel= 1
UNET Pardiso=0
UNET DZMax Abort= 0
UNET Use Existing IB Tables= 0
UNET Froude Reduction=False
UNET Froude Limit= 0
UNET Froude Power= 0
UNET D1 Cores= 0
UNET WindReference=Eulerian
UNET WindDragFormulation=Hsu (1988)
UNET D2 Coriolis=0
UNET D2 Cores= 0
UNET D2 Theta= 1
UNET D2 Theta Warmup= 1
UNET D2 Z Tol= 0.01
UNET D2 Volume Tol= 0.01
UNET D2 Max Iterations= 20
UNET D2 Equation= 0
UNET D2 RampUpFraction=0.1
UNET D2 TimeSlices= 1
UNET D2 Turbulence Formulation=Non-Conservative (original)
UNET D2 Eddy Viscosity=0.3
UNET D2 Transverse Eddy Viscosity=0.1
UNET D2 Smagorinsky Mixing=0
UNET D2 BCVolumeCheck=0
UNET D2 Cores=0
UNET D2 SolverType=PARDISO (Direct)
UNET D2 Minimum Iterations= 2147483647
UNET D2 Maximum Iterations= 2147483647
UNET D2 Restart Number= 10
UNET D2 Relaxation Coeff=1.3
UNET D2 SOR Precondition Iterations= 10
UNET D2 ILUT Maximum Fill= 8
UNET D2 ILUT Tolerance=1E-08
UNET D1D2 MaxIter= 0
UNET D1D2 ZTol=0.01
UNET D1D2 QTol=0.1
UNET D1D2 MinQTol=1
DSS File=dss
Write IC File= 0
Write IC File at Fixed DateTime=0
Write IC File at Sim End=0
Echo Input=False
Echo Parameters=False
Echo Output=False
Write Detailed= 0
HDF Write Warmup=0
HDF Write Time Slices=0
HDF Flush=0
HDF Compression= 1
HDF Chunk Size= 1
HDF Spatial Parts= 1
HDF Use Max Rows=0
HDF Fixed Rows= 1
Calibration Method= 0
Calibration Iterations= 20
Calibration Max Change=0.05
Calibration Tolerance=0.2
Calibration Maximum=1.5
Calibration Minimum=0.5
Calibration Optimization Method= 1
WQ AD Non Conservative
WQ ULTIMATE=-1
WQ Max Comp Step=1HOUR
WQ Output Interval=15MIN
WQ Output Selected Increments= 0
WQ Output face flow=0
WQ Output face velocity=0
WQ Output face area=0
WQ Output face dispersion=0
WQ Output cell volume=0
WQ Output cell surface area=0
WQ Output cell continuity=0
WQ Output cumulative cell continuity=0
WQ Output face conc=0
WQ Output face dconc_dx=0
WQ Output face courant=0
WQ Output face peclet=0
WQ Output face adv mass=0
WQ Output face disp mass=0
WQ Output cell mass=0
WQ Output cell source sink temp=0
WQ Output nsm pathways=0
WQ Output nsm derived pathways=0
WQ Create Restart=0
WQ Fixed Restart=0
WQ System Summary=0
WQ Write To DSS=0
Sorting and Armoring Iterations= 10
XS Update Threshold= 0.02
Bed Roughness Predictor= 0
Hydraulics Update Threshold= 0.02
Energy Slope Method= 1
Volume Change Method= 1
Sediment Retention Method= 0
Sediment TS Multiplier= 1
Warm Up Method= 0
XS Weighting Method= 0
Number of US Weighted Cross Sections= 1
Number of DS Weighted Cross Sections= 1
Upstream XS Weight=0
Main XS Weight=1
Downstream XS Weight=0
Number of DS XS's Weighted with US Boundary= 1
Upstream Boundary Weight= 1
Weight of XSs Associated with US Boundary= 0
Number of US XS's Weighted with DS Boundary= 1
Downstream Boundary Weight= 0.5
Weight of XSs Associated with DS Boundary= 0.5
Percentile Method= 0
Sediment Output Level= 3
Mass or Volume Output= 0
Output Increment Type= 1
Profile and TS Output Increment= 1
Transport Output Increment 1
XS Output Flag= 0
XS Output Increment= 10
Read HDF5 Sediment Hotstart= 0
Sediment Hotstart Type= 0
Write Gradation File= 0
Read Gradation Hotstart= 0
Write HDF5 File= 1
Write Binary Output= 1
Write DSS Sediment File= 0
DSS Sediment Output Type= 1
SV Curve= 0
Specific Gage Flag= 0
Subcell Erosion Methods= 0
Subcell Deposition Methods= 0
Advection Scheme= 1
Matrix Solver= 0
Implicit Weighting Factor= 1
Maximum Outer Loop Convergence Iterations= 5
Convergence Maximum Absolute= 0.001
Convergence RMSE= 0.0001
Grain Fractions Max Abs Error= 0.001
Max Subgrid Regions= 1
Max Subgrid Length Scale= 3.402823E+38
Initial Layer Thickness= 3.402823E+38
Min Layer Thickness= 3.402823E+38
Max Layer Thickness= 3.402823E+38
Number of Layers= 5

--- GLADERN.f01 (steady flow) ---

Flow Title=Flow
Program Version=6.10
Number of Profiles= 6
Profile Names=01pct,10pct,04pct,02pct,0_2pct,01plus
River Rch & RM=GLADERN,Main            ,5925
     541     285     380     458     756     800
River Rch & RM=GLADERN,Main            ,3939
     602     319     424     510     840     891
Boundary for River Rch & Prof#=GLADERN,Main            , 1
Up Type= 0
Dn Type= 3
Dn Slope=0.04598
Boundary for River Rch & Prof#=GLADERN,Main            , 2
Up Type= 0
Dn Type= 3
Dn Slope=0.04598
Boundary for River Rch & Prof#=GLADERN,Main            , 3
Up Type= 0
Dn Type= 3
Dn Slope=0.04598
Boundary for River Rch & Prof#=GLADERN,Main            , 4
Up Type= 0
Dn Type= 3
Dn Slope=0.04598
Boundary for River Rch & Prof#=GLADERN,Main            , 5
Up Type= 0
Dn Type= 3
Dn Slope=0.04598
Boundary for River Rch & Prof#=GLADERN,Main            , 6
Up Type= 0
Dn Type= 3
Dn Slope=0.04598
DSS Import GetInterval= 0
DSS Import GetPeak= 0
DSS Import FillOption= 0

--- GLADERN.g01 (geometry) ---

Geom Title=Geometry
Program Version=6.10

River Reach=GLADERN         ,Main
Reach XY= 30
     2260151.375       489061.08     2260051.797      488852.898
     2260187.708      488379.352     2260269.825      488367.661
     2260417.378      488198.085     2260586.522      488116.723
     2260729.291      487889.533     2260934.407      487834.612
     2261125.336      487947.528     2261546.116      487940.884
     2261669.917      487984.459     2261715.307      488086.603
     2261778.881      488062.647       2261775.9       487951.52
     2261862.716      487919.751     2261981.114      488024.458
     2262112.615      487986.435     2262100.206      488174.005
     2262154.709      488207.099     2262425.445      488160.027
     2262474.087      488106.382     2262722.336      488148.364
     2262907.654      488095.8882263003.19879738488004.367452897
     2263082.255      488023.145     2263154.736      487898.435
       2263381.9      487841.976      2263439.09       487517.53
     2263624.245      487196.997     2263730.173      487104.345

Type RM Length L Ch R = 1 ,5925    ,160.3,167.3,172.4
XS GIS Cut Line= 3
2260308.04476798488962.7018051562260266.86733812 488973.44609046
2260041.33569587489132.267477017
#Sta/Elev= 30
       0 2382.09       4 2379.54     8.1 2377.55    32.9 2366.28    37.1 2363.71
    45.8  2356.9    47.2 2356.42    61.5 2357.08      73 2356.54    75.9 2355.89
    81.6 2352.93    90.2 2349.63   110.3 2346.68   146.3  2346.7   167.7 2346.13
   182.22345.196   187.7  2344.5   192.6 2344.68     1972345.566   201.9 2346.23
   212.2 2346.68   226.9 2348.83   242.4 2350.08   246.4 2352.29   251.3 2356.04
   265.3 2364.29   285.6 2374.96   302.7 2385.02   314.1 2392.97   318.4  2394.1
#Mann= 5 ,-1,0
       0      .1       0      30     .06       0  142.56      .1       0
   182.2    .045       0     197      .1       0
Bank Sta=182.2,197
XS Rating Curve= 0 ,0
Exp/Cntr=0.3,0.1

Type RM Length L Ch R = 1 ,5758    ,68.3,75.1,82.1
XS GIS Cut Line= 4
2260291.73599066488929.0081751012260105.30745475488913.301741672
2260023.36084555488924.9108446412259974.87576845 488937.88572443
#Sta/Elev= 30
       0    2376    15.6 2368.77    31.7 2363.22    43.7 2353.65    47.7 2351.77
    51.7 2350.79    71.8 2351.02    99.9 2349.34     116  2349.5     128 2345.65
   140.1 2344.71   180.2 2343.86     188    2344   200.4 2345.11   204.4 2344.83
   209.2 2343.61   221.5 2342.94   228.6 2342.34   232.7 2342.52   235.6  2343.3
   248.8 2345.54     269 2346.93   273.2 2349.89   277.3 2354.32   281.4 2357.62
     298 2368.55   306.3 2375.89   310.4 2378.23   318.7 2379.69     320 2380.94
#Mann= 5 ,-1,0
       0      .1       0      10     .06       0     110      .1       0
   221.5    .045       0   235.6      .1       0
Bank Sta=221.5,235.6
XS Rating Curve= 0 ,0
Exp/Cntr(USF)=0,0
Exp/Cntr=0.5,0.3

Type RM Length L Ch R = 1 ,5683    ,52.3,52.6,55
XS GIS Cut Line= 5
2260290.37148352488919.6253216182260145.00973834488907.830461606
2260079.15087962 488861.789171882260001.50841643 488815.64869905
2259948.24312046 488821.79469474
#Sta/Elev= 30
       0 2375.41    10.2 2370.66    18.3 2367.23    30.3 2363.19    34.7 2360.77
    46.3 2351.58    50.4 2350.54    54.4  2349.8      74 2350.35   110.6 2348.72
   118.6 2348.93   130.6    2346   134.6 2345.92   145.8  2344.5   176.1 2343.43
   217.3 2343.18   240.5 2343.01250.59852342.257   257.6 2341.45262.56012342.095
   266.9 2342.37   276.2  2341.5   285.5 2345.15   290.1 2345.59   308.8 2345.26
   313.5  2346.4   316.5 2347.49   337.1 2357.74   351.6 2362.25   370.1 2371.92
#Mann= 7 ,-1,0
       0      .1       0    10.2     .06       0   110.6      .1       0
   176.1     .06       0   217.3      .1       0250.5985    .045       0
262.5601      .1       0
#XS Ineff= 2 , 0
          236.85    2345  280.62         2344.29
Permanent Ineff=
       F       F
Bank Sta=250.5985,262.5601
XS Rating Curve= 0 ,0
Exp/Cntr(USF)=0,0
Exp/Cntr=0.5,0.3

Type RM Length L Ch R = 1 ,5630    ,80,80,75.8
XS GIS Cut Line= 5
2260305.39375886488850.4760079572260131.25721432488835.452462938
2260032.23839488488773.9878128442259993.96891282488750.769893042
2259923.50941906488782.710950334
#Sta/Elev= 30
       0 2371.61    29.3  2365.5    31.9 2364.57    37.4 2361.32    45.4 2353.27
    49.4 2351.23    57.4 2349.18    89.6 2349.14   129.7 2347.12   161.8  2343.6
   178.4 2343.88     202 2342.68   211.4  2343.1   234.9 2341.63   244.3 2339.39
   254.9 2338.85262.08222339.167   265.8 2339.62   272.6 2339.99   277.3 2339.52
   296.1 2339.37   300.7 2340.02   310.1 2340.16   342.5 2342.51   360.4 2345.47
   378.6 2345.52   381.6 2346.24   390.6 2352.54   408.3 2357.56   413.5 2360.18
#Mann= 5 ,-1,0
       0     .06       0   234.9      .1       0   244.3    .045       0
262.0822      .1       0   265.8     .06       0
#XS Ineff= 2 ,-1
    3.25  239.25    2343  268.59  392.392341.624
Permanent Ineff=
       F       F
Bank Sta=244.3,262.0822
XS Rating Curve= 0 ,0
Exp/Cntr(USF)=0,0
Exp/Cntr=0.5,0.3

Type RM Length L Ch R = 1 ,5550    ,115.4,110.1,105.2
XS GIS Cut Line= 4
2260297.88198635 488821.111806332260025.31552385488693.284692439
2259943.62197099488652.8122562032259867.20374576488693.355355279
#Sta/Elev= 30
       0 2359.19     7.2 2355.03    10.7 2353.67    15.1  2353.1    32.8 2352.84
    43.3 2352.17    46.9 2351.52    56.4  2348.2    64.4 2346.67    72.6  2346.4
   107.9 2344.27   138.8 2341.36   172.7 2340.42   205.1 2340.46   214.8 2339.14
   223.8 2338.85   228.52337.977   231.6 2337.22   235.4 2336.99   240.5 2337.21
     245 2338.06   250.9 2339.67   253.9    2340   301.1 2339.93   342.5 2340.26
   379.6  2342.3   392.2 2342.46   410.1 2343.35   459.5  2344.3   478.7 2345.64
#Mann= 5 ,-1,0
       0     .06       0    72.6     .05       0   228.5    .045       0
     245     .06       0   301.1     .05       0
#XS Ineff= 2 , 0
          196.97 2343.98
Permanent Ineff=
       F       F
Bank Sta=228.5,245
XS Rating Curve= 0 ,0
Exp/Cntr(USF)=0,0
Exp/Cntr=0.3,0.1

Type RM Length L Ch R = 1 ,5440    ,133.7,140.8,147.3
XS GIS Cut Line= 5
2260292.98361896488799.8525980232260197.20638304488667.380034374
2260139.53724466488625.4497878122260100.81456498488624.167410365
2259942.69843906488542.083013669
#Sta/Elev= 30
       0 2354.24     8.2 2354.28    11.1 2353.91      14 2353.29      23 2349.54
      28 2348.36    42.8 2347.08    54.1 2345.45    91.3 2343.78   119.9 2340.35
   134.3 2339.38   194.4 2337.69   214.5 2337.58   238.1 2338.16   242.2 2337.52
   246.1 2335.51 247.4932335.357   254.1 2334.83   258.7 2335.28   262.1 2335.74
   270.2 2337.92   274.2 2338.18   278.7 2337.78   287.8 2337.92   310.3 2337.41
   355.4 2337.37   368.9  2337.9   403.8 2340.28     423 2340.45   451.7 2340.08
#Mann= 4 ,-1,0
       0     .06       0    11.1     .05       0 247.493    .045       0
   258.7     .05       0
Bank Sta=247.493,258.7
XS Rating Curve= 0 ,0
Exp/Cntr=0.3,0.1

Type RM Length L Ch R = 1 ,5299    ,49.4,47.6,46
XS GIS Cut Line= 3
2260334.29193635488612.3625914922260064.79601996488440.455725607
2259883.13024902488482.494085823
#Sta/Elev= 30
       0 2338.83    21.5 2338.26    65.4 2335.55    73.4 2335.31    97.4 2335.19
   135.4 2334.69   147.2 2334.92   159.1 2335.43   171.8  2335.2   191.9 2335.56
   200.8 2335.22   211.3 2335.46   215.3 2334.89   220.8 2333.46     224 2333.19
   232.3 2332.97   238.5  2333.1   244.3 2333.49   249.2 2334.66     254 2335.05
   267.4 2334.59   291.9 2335.35   320.8 2335.96   344.9 2337.09   377.8 2337.59
   410.3 2338.43   444.1 2338.25   460.8 2338.49   484.5 2339.38   506.1 2339.95
#Mann= 3 ,-1,0
       0     .05       0   220.8    .045       0   244.3     .05       0
#XS Ineff= 2 , 0
           98.55 2338.11  254.11         2338.01
Permanent Ineff=
       F       F
Bank Sta=220.8,244.3
XS Rating Curve= 0 ,0
Exp/Cntr(USF)=0,0
Exp/Cntr=0.3,0.1

Type RM Length L Ch R = 1 ,5252    ,192.2,197.4,201.2
XS GIS Cut Line= 2
 2260416.3663694488563.7447443512259974.01371855488359.742110075
#Sta/Elev= 30
       0 2338.56    44.3  2338.5    57.5 2337.91    79.5 2335.81   101.5 2334.53
   119.6 2334.38   146.8 2333.69     189 2333.77     198 2333.96   215.9 2333.44
   229.3 2333.52   242.5 2334.31   252.3 2335.52   258.3 2335.67   260.1 2335.59
   264.5 2334.81   270.4 2333.01   273.3 2332.11   277.7 2331.82   282.1    2332
   285.5 2332.89   290.9 2334.44   295.3 2334.66   299.7 2334.64   308.6 2333.91
   311.8 2333.91   369.9 2335.62     400 2336.83   458.3 2337.55   487.1  2337.4
#Mann= 3 ,-1,0
       0     .05       0   270.4    .045       0   285.5     .05       0
#XS Ineff= 2 , 0
          121.05 2336.22  298.78         2336.16
Permanent Ineff=
       F       F
Bank Sta=270.4,285.5
XS Rating Curve= 0 ,0
Exp/Cntr(USF)=0,0
Exp/Cntr=0.3,0.1

Type RM Length L Ch R = 1 ,5054    ,171.8,171.1,169.8
XS GIS Cut Line= 3
2260424.27410568488493.1790561182260396.68055209488433.470121834
 2260101.8944326488170.336792033
#Sta/Elev= 30
       0  2337.4    47.9  2336.7    60.3 2336.12    77.2 2334.85   108.8 2331.88
   114.5 2331.56   138.3 2331.17   146.9 2331.23   157.6 2331.73   179.1 2331.46
   188.2 2329.52   192.4 2328.78   196.7 2328.71  201.312329.352   205.2 2330.06
   216.5 2330.16   222.4  2331.4   227.8 2332.21   230.7 2332.32   240.4  2331.9
   243.4 2331.95   248.8 2332.56   259.5 2332.73   270.2 2332.13   307.7 2331.88
   342.5 2332.52   388.2  2332.7   402.6 2333.15   436.4  2335.3   460.9 2335.65
#Mann= 3 ,-1,0
       0     .05       0   188.2    .045       0  201.31     .05       0
#XS Ineff= 2 , 0
                          231.83         2333.18
Permanent Ineff=
       F       F
Bank Sta=188.2,201.31
XS Rating Curve= 0 ,0
Exp/Cntr(USF)=0,0
Exp/Cntr=0.3,0.1

Type RM Length L Ch R = 1 ,4883    ,224.2,227.8,228
XS GIS Cut Line= 2
2260599.95460553 488355.720138262260203.71071334488073.759354456
#Sta/Elev= 30
       0 2331.26      39 2330.94    61.9 2331.23    79.1 2331.05   107.9 2331.28
   122.5 2330.51   142.2 2328.76   151.9 2328.17   156.6 2328.06   176.6  2328.8
   186.3 2329.55   196.1 2328.53   205.9 2328.84   213.9 2327.96   225.2 2327.95
     234 2327.46   240.3 2326.93   245.2 2327.57   248.3 2328.35     255 2329.28
   266.6 2329.03   279.9 2328.11   287.2 2328.12   294.1 2328.59   323.7  2329.5
   363.1 2329.59   425.2 2330.58   446.3  2331.4   474.9 2333.19   486.3 2333.63
#Mann= 5 ,-1,0
       0     .05       0     150     .07       0     234    .045       0
   245.2     .07       0     270     .05       0
#XS Ineff= 2 , 0
                          305.96         2331.39
Permanent Ineff=
       F       F
Bank Sta=234,245.2
XS Rating Curve= 0 ,0
Exp/Cntr(USF)=0,0
Exp/Cntr=0.3,0.1

Type RM Length L Ch R = 1 ,4655    ,161.5,162,162.6
XS GIS Cut Line= 4
2260656.05992246488243.1049052132260646.68347669488161.907104135
2260408.19085096487938.2780414832260307.45744711 487912.55199547
#Sta/Elev= 30
       0 2329.03    22.1 2328.74    50.3    2329    70.2 2328.75    92.5 2328.13
   117.9 2326.13   141.3 2325.81     151 2326.12155.40352325.692   157.6 2325.52
163.23922325.648   170.5 2326.05   177.4 2326.06   185.9 2325.82   194.8 2326.42
   197.2 2326.43   214.2 2326.06   223.2 2326.22   244.2 2326.07   258.2 2326.27
   269.9 2326.23   281.6 2325.82   293.3 2326.16   381.2 2327.12   403.2 2327.56
   449.1 2329.12   462.4 2330.01     483  2331.7   503.6 2332.91   512.6 2333.19
#Mann= 5 ,-1,0
       0     .05       0155.4035    .045       0163.2392     .05       0
  171.74     .07       0  311.74     .05       0
#XS Ineff= 2 , 0
                          336.88         2328.51
Permanent Ineff=
       F       F
Bank Sta=155.4035,163.2392
XS Rating Curve= 0 ,0
Exp/Cntr(USF)=0,0
Exp/Cntr=0.3,0.1

Type RM Length L Ch R = 1 ,4493    ,236.3,247.4,254.4
XS GIS Cut Line= 4
2260698.67415764488185.4057150262260709.43448564488006.522664366
2260584.41087774 487891.086574662260364.67807166487889.850778142
#Sta/Elev= 30
       0 2328.75    60.3 2327.48    76.4 2326.62    88.4 2326.32   108.4 2324.55
   124.5 2324.09   164.5 2324.83   168.5 2324.55   186.4 2324.45  216.83 2324.65
  238.64 2324.68   251.9 2325.43     283  2324.6   302.8 2325.03   328.6 2324.67
   346.3  2325.3   349.6 2325.16   385.6 2325.77   393.6 2326.48   401.6  2326.4
   409.6 2326.73   433.6 2326.36   441.6 2326.51   449.6 2326.21   453.6 2326.61
   465.6 2326.88   529.6 2327.89   541.6 2328.77   557.6 2329.33   569.1 2330.38
#Mann= 5 ,-1,0
       0     .05       0  189.21      .1       0  216.83    .045       0
  238.64     .08       0  329.21      .1       0
#XS Ineff= 2 , 0
                           337.2         2326.66
Permanent Ineff=
       F       F
Bank Sta=216.83,238.64
XS Rating Curve= 0 ,0
Exp/Cntr(USF)=0,0
Exp/Cntr=0.3,0.1

Type RM Length L Ch R = 1 ,4246    ,84.9,85.2,85.6
XS GIS Cut Line= 4
2260829.07021739488142.4572300242260855.76734195488089.062980905
2260849.10863413487790.0189158872260834.09493405487744.977815655
#Sta/Elev= 30
       0 2324.89    14.8 2323.99    23.8 2324.18      42 2323.19    51.7 2323.35
    70.9  2322.6   103.6  2322.7   119.6 2322.24   143.6 2322.29   151.6 2322.01
   163.6 2322.49   223.6 2322.44   243.6 2322.74   247.6  2322.6   251.6 2321.95
   263.6 2322.16   295.6 2322.05   305.42321.386   311.6 2320.95   319.12321.335
   327.6  2322.5   331.6 2323.93   339.6 2330.63   343.7 2333.71   347.7 2336.42
   351.7 2338.63     365 2340.71   380.8 2342.62   393.4 2343.78   406.3 2346.32
#Mann= 4 ,-1,0
       0     .05       0   249.7      .1       0   305.4    .045       0
   319.1      .1       0
#XS Ineff= 2 , 0
           82.23 2327.61
Permanent Ineff=
       F       F
Bank Sta=305.4,319.1
XS Rating Curve= 0 ,0
Exp/Cntr(USF)=0,0
Exp/Cntr=0.3,0.1

Type RM Length L Ch R = 1 ,4161    ,220.6,222,222.2
XS GIS Cut Line= 3
 2260901.6565844488179.6244328942260933.18535456488108.309357526
2260936.00184552487740.771686732
#Sta/Elev= 30
       0 2324.79    61.4 2323.59   101.1 2323.42   119.8 2322.24   161.1 2321.56
   185.1 2321.78   201.1 2321.39   221.1 2321.74   237.1 2321.51   249.1 2322.01
   291.8 2321.28   317.1  2322.2   329.1 2321.05   337.1 2321.18   345.7 2319.79
   352.2 2319.59   359.42320.032   361.9 2320.37   365.1 2321.54   368.3 2326.18
   373.1 2331.96   377.1 2335.58   381.1 2337.91   385.1 2338.83   393.1 2339.99
   401.1 2340.24   409.1 2340.93   425.1 2342.99   433.4 2345.11   445.5 2348.99
#Mann= 4 ,-1,0
       0     .05       0  287.97      .1       0   345.7    .045       0
   359.4      .1       0
#XS Ineff= 2 , 0
          136.07 2326.79
Permanent Ineff=
       F       F
Bank Sta=345.7,359.4
XS Rating Curve= 0 ,0
Exp/Cntr(USF)=0,0
Exp/Cntr=0.3,0.1

Type RM Length L Ch R = 1 ,3939    ,148.6,144.3,139.7
XS GIS Cut Line= 3
2261056.30333249488193.669641765 2261104.3581567488115.866593048
2261136.39470617487819.528510437
#Sta/Elev= 30
       0 2323.65    52.6 2323.14    91.1 2321.93   118.3  2321.9   134.4 2321.04
   142.4 2320.29   166.6 2320.37   178.6 2320.97   198.4 2320.97   206.3 2320.61
   214.8 2320.83   218.9 2320.46   226.9  2320.4     239 2320.53     243 2320.12
   248.1  2318.9   251.1 2318.44   255.1 2318.39   263.1  2318.6  265.09 2318.95
   271.2 2319.84   283.2 2320.81   299.3 2320.47   303.4 2320.61   307.4 2321.55
   315.4 2326.84   319.5 2327.85   347.9 2331.58   363.7 2334.16   389.5 2336.73
#Mann= 4 ,-1,0
       0     .05       0  211.45      .1       0   248.1    .045       0
  265.09      .1       0
#XS Ineff= 2 , 0
           121.1 2324.57
Permanent Ineff=
       F       F
Bank Sta=248.1,265.09
XS Rating Curve= 0 ,0
Exp/Cntr(USF)=0,0
Exp/Cntr=0.3,0.1

Type RM Length L Ch R = 1 ,3794    ,93.6,101.4,108.6
XS GIS Cut Line= 5
2261175.78930394 488189.092991842261245.15715342488133.747130885
2261269.29890373487953.3284728072261261.04136869487932.309292699
2261270.80027374487808.446267061
#Sta/Elev= 30
       0 2322.76      64 2322.09   101.4 2320.83   129.7 2320.75   149.8 2319.95
   190.2 2319.21   214.4 2319.34   226.5 2319.89   266.9  2319.8   270.8 2319.14
   273.8 2318.18   275.2 2317.78   279.5 2317.48   287.2 2318.32   292.4 2318.95
   296.5 2319.03   304.5  2317.9   308.5  2317.7   328.6 2317.75   332.6 2318.13
   336.6 2319.59   344.6 2323.72   348.7 2326.98   352.7 2330.91   368.7 2332.89
   388.8 2334.22   396.8 2335.14   408.8 2336.96   412.9 2338.14   417.6 2338.84
#Mann= 4 ,-1,0
       0     .05       0  218.74      .1       0   273.8    .045       0
   287.2      .1       0
#XS Ineff= 2 , 0
          136.07 2324.49  319.65         2324.66
Permanent Ineff=
       F       F
Bank Sta=273.8,287.2
XS Rating Curve= 0 ,0
Exp/Cntr(USF)=0,0
Exp/Cntr=0.3,0.1

Type RM Length L Ch R = 1 ,3693    ,76.8,74.4,72.4
XS GIS Cut Line= 4
2261297.85186316488218.1639083492261306.47833736488092.739825738
2261366.67576783487910.3233697992261373.36437121487848.301774779
#Sta/Elev= 30
       0 2322.03    49.1 2321.72    57.1  2321.4    65.1 2321.41    85.6 2320.85
   129.5 2321.02   150.5 2320.11   177.4 2319.83   196.4 2319.86   201.1 2320.04
   205.3 2319.81   213.7 2318.86   217.9 2318.74   229.2 2319.28     239 2319.19
   247.4 2318.66   251.6  2318.7   255.8 2319.13   264.3 2319.15   272.4 2317.72
   281.9 2317.53  290.34 2317.72   293.7 2318.19   302.2  2322.4   307.2 2324.36
   314.8 2326.62     327 2328.79   351.1 2329.92   371.3 2331.61   380.2 2332.64
#Mann= 4 ,-1,0
       0     .05       0  225.72      .1       0   272.4    .045       0
  290.34      .1       0
#XS Ineff= 2 , 0
          128.18 2323.53
Permanent Ineff=
       F       F
Bank Sta=272.4,290.34
XS Rating Curve= 0 ,0
Exp/Cntr(USF)=0,0
Exp/Cntr=0.3,0.1

Type RM Length L Ch R = 1 ,3619    ,205.1,207,206.1
XS GIS Cut Line= 2
2261387.58910976488233.8028258252261445.41298569487834.818081916
#Sta/Elev= 30
       0 2322.07    24.9 2321.48    49.1 2321.57    77.4 2320.23    85.5 2320.66
    89.5 2320.61   142.3 2318.34   154.2 2318.27   178.5 2318.89   194.6 2318.24
   210.8 2318.92   222.9 2318.88     231 2319.19   243.1 2319.11   251.2 2319.36
   259.3 2318.85   263.3 2317.86   271.4 2317.53     280  2317.7   287.6 2318.84
   294.1 2319.19   299.7 2319.95   303.8 2320.87   315.9 2324.52   319.9 2325.46
     324 2326.09   329.4 2326.41   344.2 2328.86   396.7 2334.38   403.2 2335.45
#Mann= 5 ,-1,0
       0     .08       0      40     .05       0     240      .1       0
   263.3    .045       0     280      .1       0
#XS Ineff= 2 , 0
          115.94 2323.78
Permanent Ineff=
       F       F
Bank Sta=263.3,280
XS Rating Curve= 0 ,0
Exp/Cntr(USF)=0,0
Exp/Cntr=0.3,0.1

Type RM Length L Ch R = 1 ,3412    ,188.2,192.4,180.9
XS GIS Cut Line= 2
2261553.27600491488313.3320689552261643.28628912487870.321941737
#Sta/Elev= 30
       0  2321.7    28.7 2321.55    36.9 2321.21    45.1 2321.33    80.6 2320.55
   138.3  2320.2   151.9 2319.75   171.6 2319.52   200.2 2318.33     241 2317.71
     290 2318.44   298.1 2318.35   306.3 2317.89   318.1 2317.96   326.7 2318.49
   338.9  2318.6   347.1 2318.26  350.082317.611   355.3 2317.05   363.4 2317.71
   367.5    2318   371.6 2318.69   375.8 2320.23   379.8 2322.15   387.9 2325.16
     392    2327   400.2 2329.06   416.5 2331.21     441 2334.95   452.1 2335.64
#Mann= 5 ,-1,0
       0     .05       0     220     .07       0     320      .1       0
  350.08    .045       0   363.4      .1       0
#XS Ineff= 2 , 0
          135.27 2325.11
Permanent Ineff=
       F       F
Bank Sta=350.08,363.4
XS Rating Curve= 0 ,0
Exp/Cntr(USF)=0,0
Exp/Cntr=0.3,0.1

Type RM Length L Ch R = 1 ,3219    ,289.4,292.9,283.3
XS GIS Cut Line= 2
2261700.62445986488355.8672505742261749.56657307487881.655421419
#Sta/Elev= 30
       0    2321    26.8 2321.28    38.9 2320.86      55 2320.95      63 2320.63
    71.3 2320.74    87.1 2320.37   118.7 2320.87   151.5 2319.69   173.4 2319.78
   187.4  2320.1   235.9 2320.26     244 2319.87  266.45 2317.29   272.1 2316.81
   280.2 2316.88   282.7 2317.29   292.2  2318.2   296.3 2318.34   332.4 2317.89
   348.5 2318.24   400.8 2317.94   416.9 2318.15     425 2317.94     429 2318.25
     445 2326.82   453.1 2330.73   457.1 2332.11   461.1 2332.92   476.7 2334.81
#Mann= 4 ,-1,0
       0     .07       0  266.45    .045       0   282.7     .07       0
     360      .1       0
#XS Ineff= 2 , 0
          226.74  2324.9
Permanent Ineff=
       F       F
Bank Sta=266.45,282.7
XS Rating Curve= 0 ,0
Exp/Cntr(USF)=0,0
Exp/Cntr=0.3,0.1

Type RM Length L Ch R = 1 ,2926    ,152,155.6,156.9
XS GIS Cut Line= 2
2261805.29889438488353.7624768692261881.75195344487862.920485618
#Sta/Elev= 30
       0 2320.73    45.1 2319.94    61.3  2319.4    69.4 2319.85    85.6  2319.7
   146.3 2318.36   275.9 2317.92     288  2317.8   293.8  2317.5   320.4  2317.5
   336.6 2316.91   346.3 2317.39   360.9 2317.24   377.1 2317.61   385.2 2317.35
   419.8 2317.57   428.8  2316.9   433.6 2316.81   441.8 2316.88   445.9  2316.9
   449.9 2317.84   454.9 2321.95     458 2323.79   466.1 2324.69   470.2 2325.95
   474.2 2328.09   478.3 2329.62   486.4 2331.81   494.5 2333.57   496.8 2333.79
#Mann= 6 ,-1,0
       0     .05       0      60     .07       0     260     .05       0
     360      .1       0   428.8    .045       0   441.8      .1       0
#XS Ineff= 2 , 0
          151.99 2321.22
Permanent Ineff=
       F       F
Bank Sta=428.8,441.8
XS Rating Curve= 0 ,0
Exp/Cntr(USF)=0,0
Exp/Cntr=0.3,0.1

Type RM Length L Ch R = 1 ,2771    ,406.3,403.4,401.1
XS GIS Cut Line= 2
2261874.41991673488345.5548104812262029.54978032487889.982059552
#Sta/Elev= 30
       0 2319.88    21.5 2319.93    63.8 2319.18    68.3 2319.31   101.8 2318.31
   152.5 2317.63   190.5 2317.32     199 2317.48   232.8 2316.98   258.2 2317.22
   283.5 2317.04   296.2 2317.52   313.7 2317.01   326.4 2317.17   332.7 2316.96
     339 2316.81  348.24 2316.93   359.6 2317.59   389.1 2316.91   405.2 2317.09
   418.7 2316.85     423 2317.07   427.4  2318.2   431.4  2320.1   435.6 2322.65
   439.8 2324.71   444.1 2325.13   455.6  2327.1   474.5 2328.86   481.3 2330.02
#Mann= 5 ,-1,0
       0     .05       0     160     .07       0     260      .1       0
   332.7    .045       0  348.24      .1       0
#XS Ineff= 2 , 0
          123.99 2321.73
Permanent Ineff=
       F       F
Bank Sta=332.7,348.24
XS Rating Curve= 0 ,0
Exp/Cntr(USF)=0,0
Exp/Cntr=0.3,0.1

Type RM Length L Ch R = 1 ,2367    ,153.4,153.2,151.2
XS GIS Cut Line= 4
2262028.54782666488403.7644368142262115.66435797488327.769164818
2262149.95490753488071.9802005372262207.41474733487916.282570105
#Sta/Elev= 30
       0 2318.83      10 2318.85   130.3 2317.79   166.6 2316.84   182.8 2316.02
   186.8  2316.1   190.9 2316.85   194.9 2317.14     203  2316.6     211 2314.97
   227.2 2315.67     2412314.499   247.4 2313.78   251.4 2314.04   253.6 2314.58
   263.5 2316.19   271.6 2315.77   299.9 2315.75   324.8 2316.72   352.3 2316.67
   372.5  2317.9   421.2 2317.77   449.2  2318.5   457.7  2319.3     471 2319.93
   487.5 2322.14   492.8 2322.47   513.1 2325.35   530.2 2327.34   539.6 2328.85
#Mann= 6 ,-1,0
       0     .05       0      10     .07       0      40     .05       0
     241    .045       0   253.6     .07       0  453.68      .1       0
#XS Ineff= 2 , 0
           194.2 2319.47
Permanent Ineff=
       F       F
Bank Sta=241,253.6
XS Rating Curve= 0 ,0
Exp/Cntr(USF)=0,0
Exp/Cntr=0.3,0.1

Type RM Length L Ch R = 1 ,2214    ,108.8,107.5,106.6
XS GIS Cut Line= 3
2262182.39191387488423.2266406182262252.82655621488299.966016526
2262283.41001933487957.987292542
#Sta/Elev= 30
       0 2318.82   117.1 2317.43   180.8 2315.63     193 2314.78   210.3 2315.69
   217.1 2315.28   221.1 2314.38     225 2313.97   241.1 2314.74   249.2 2314.87
   273.3 2314.75   277.3 2314.16   281.3 2313.78   285.3 2313.89   286.62314.156
   289.3 2314.71   293.4 2315.08   309.4 2315.05   313.5 2314.78   333.5 2315.62
   341.5 2315.42   353.6 2315.59   369.7 2315.19   389.7  2315.1   397.8 2315.42
   410.4 2316.97   429.9  2319.9   437.9 2320.45   449.9 2322.27   485.3 2325.91
#Mann= 5 ,-1,0
       0     .05       0  241.97     .07       0   277.3    .045       0
   286.6     .07       0  441.97      .1       0
#XS Ineff= 2 , 0
          209.34 2318.83
Permanent Ineff=
       F       F
Bank Sta=277.3,286.6
XS Rating Curve= 0 ,0
Exp/Cntr(USF)=0,0
Exp/Cntr=0.3,0.1

Type RM Length L Ch R = 1 ,2107    ,131.1,126.8,122.2
XS GIS Cut Line= 3
2262449.30213747488349.0849118412262370.52655064488225.824287749
2262367.74623581487956.133749323
#Sta/Elev= 30
       0 2319.94    80.6 2318.34    85.3 2318.44   109.1 2317.54   132.8 2317.31
   146.9 2316.21   158.9 2316.32   166.9 2315.45   178.9 2314.88   182.9 2314.53
   186.9 2313.58   191.62313.073   194.9 2312.77   202.42313.019   210.9 2314.29
   222.9 2314.43   226.9 2314.44   238.9  2313.9   250.9 2314.49   266.9 2314.07
   306.9 2314.18   322.9 2313.97   326.9 2314.12   330.9 2314.58   338.9 2317.56
   346.9 2320.01   362.9 2323.06     383 2325.19   398.7    2326     416 2327.77
#Mann= 6 ,-1,0
       0     .07       0      60     .05       0  176.28     .07       0
   191.6    .045       0   202.4     .07       0  276.28      .1       0
Bank Sta=191.6,202.4
XS Rating Curve= 0 ,0
Exp/Cntr(USF)=0,0
Exp/Cntr=0.3,0.1

Type RM Length L Ch R = 1 ,1980    ,107.5,112.2,114.9
XS GIS Cut Line= 5
2262516.02969337488331.4762512572262468.76434127488226.751059359
2262470.61788449488122.0258674612262459.49662517 488095.14949078
2262455.78953873487974.669181517
#Sta/Elev= 30
       0 2321.17    20.1 2320.67      64 2318.83    72.7 2318.97    81.5 2318.72
    98.4 2317.66   115.9 2317.04   140.5 2315.73   145.6 2314.93   152.5 2314.28
   174.1 2313.67   200.5 2313.74   208.5 2313.38   224.9 2313.28   229.2 2312.29
   233.5 2311.75   237.9 2312.17   246.5 2311.77   250.7 2312.43   265.5 2313.51
   274.7 2313.86   290.7 2315.84   302.7  2316.6   318.7 2318.81   326.7  2320.6
   334.7 2321.71   342.7 2323.25   350.9 2324.48   358.8 2325.48   369.3 2326.07
#Mann= 5 ,-1,0
       0     .05       0      40     .07       0   229.2    .045       0
   237.9     .07       0  338.73      .1       0
Bank Sta=229.2,237.9
XS Rating Curve= 0 ,0
Exp/Cntr(USF)=0,0
Exp/Cntr=0.3,0.1

Type RM Length L Ch R = 1 ,1868    ,145.3,143.5,141.5
XS GIS Cut Line= 3
 2262624.4619717488308.3069610142262561.51935106488219.414735296
2262574.41630478487980.229811175
#Sta/Elev= 30
       0 2322.58    28.3 2322.06    69.7 2320.26      97 2318.63   109.8 2317.38
   115.2 2316.62   123.2 2314.59   127.2 2314.14   135.2 2314.48   139.2 2314.29
   143.2 2313.81   147.2 2312.76   151.2 2312.42   175.3 2312.87   179.3 2312.83
   183.3 2312.51   203.3 2312.66   210.1 2311.85   215.3 2311.18   219.3 2311.23
  221.84 2311.76   223.3 2312.11     239 2313.76   246.6  2315.1   255.4 2316.34
   303.4 2321.31   307.4 2321.97   315.5 2322.67   323.5 2323.95   348.5 2326.52
#Mann= 6 ,-1,0
       0     .05       0  128.92     .07       0   210.1    .045       0
  221.84     .07       0  228.92     .05       0  328.92      .1       0
#XS Ineff= 2 , 0
          136.39 2316.83
Permanent Ineff=
       F       F
Bank Sta=210.1,221.84
XS Rating Curve= 0 ,0
Exp/Cntr(USF)=0,0
Exp/Cntr=0.3,0.1

Type RM Length L Ch R = 1 ,1724    ,119.4,118,116.5
XS GIS Cut Line= 3
2262683.38611065 488314.689637092262701.62775624488201.861681008
 2262673.2518631487980.259467867
#Sta/Elev= 30
       0 2323.63    13.7 2323.23    36.9 2322.04    47.3 2321.25    70.4 2319.85
    86.6 2318.61   102.8 2317.06   114.3 2316.19   135.1 2313.31   148.4 2311.99
   151.3 2311.59   157.2 2310.42   159.3 2310.02   163.4 2309.92   168.9 2310.48
   171.4 2310.92   175.5 2311.35   195.6 2311.58   207.7 2311.24   231.9 2312.42
     236 2312.88     244 2314.86   248.1 2315.56   260.2 2318.44   264.2 2318.96
   272.3 2319.43   284.4 2320.57   304.5  2322.8   316.6 2324.52   337.7 2326.69
#Mann= 4 ,-1,0
       0     .05       0   157.2    .045       0   168.9     .05       0
  214.29      .1       0
Bank Sta=157.2,168.9
XS Rating Curve= 0 ,0
Exp/Cntr(USF)=0,0
Exp/Cntr=0.3,0.1

Type RM Length L Ch R = 1 ,1606    ,113.6,112.1,109.8
XS GIS Cut Line= 4
2262769.86502309488305.9066225452262822.56311037488185.646884925
2262786.75543568488050.523584229 2262732.7061154487995.123030943
#Sta/Elev= 30
       0 2323.92     9.5  2323.1    18.3  2322.8    35.7 2320.69    53.9 2319.27
    66.3 2318.01      75 2317.88    83.8 2317.17    92.5 2317.09   101.2 2315.72
     110 2313.41   114.3 2312.66   118.7 2312.34   144.2 2312.45   152.5 2311.81
   160.7 2311.62   173.2 2310.47     186 2310.33   199.1 2309.66   206.3  2309.2
  209.43 2308.69   214.5  2308.4   217.4 2308.65   239.4 2309.73   251.8 2311.65
   260.1 2312.32   279.5 2313.31   289.7 2315.82   314.9 2321.14   348.5 2325.08
#Mann= 5 ,-1,0
       0     .05       0      10     .07       0  209.43    .045       0
   217.4     .07       0  331.09      .1       0
Bank Sta=209.43,217.4
XS Rating Curve= 0 ,0
Exp/Cntr(USF)=0,0
Exp/Cntr=0.3,0.1

Type RM Length L Ch R = 1 ,1494    ,71.1,72.8,72.4
XS GIS Cut Line= 4
2262894.85407624488304.5553895382262944.84969749488166.729622827
  2262848.912154487997.8254969572262846.88530449487958.639739755
#Sta/Elev= 30
       0 2322.94    12.1 2321.91    20.6 2321.82    41.9 2318.69    46.1 2318.34
    50.4 2318.01    67.4 2317.87    84.4  2315.7     110 2313.97   146.6  2312.3
     176  2309.4   180.6 2309.97   185.2 2310.19   194.4  2309.3   203.6 2309.33
   209.9 2308.64   217.4 2308.58     222 2308.08   226.6  2307.9   229.92308.039
   235.8 2308.46   277.6 2309.01   295.6  2310.1   312.5 2311.68   327.8 2312.81
     337 2314.28   349.5 2317.77   357.7 2319.69   365.5 2321.81   380.1 2325.14
#Mann= 4 ,-1,0
       0     .05       0     110     .07       0     222    .045       0
   229.9      .1       0
#XS Ineff= 2 , 0
          171.98 2313.84
Permanent Ineff=
       F       F
Bank Sta=222,229.9
XS Rating Curve= 0 ,0
Exp/Cntr(USF)=0,0
Exp/Cntr=0.3,0.1

Type RM Length L Ch R = 1 ,1421    ,191.2,191.6,184.7
XS GIS Cut Line= 4
2263100.97277845488199.5168896422263002.95271679488149.163593737
2262987.80960046488127.5759937942262896.68596813487950.418508329
#Sta/Elev= 30
       0 2320.46     5.3 2320.25    20.2 2320.29    46.9 2318.81    55.8 2317.96
    73.6 2315.22    81.8 2314.33    88.5 2313.33   112.2 2311.22     122 2310.62
     141 2309.91   157.3 2309.02   179.7 2308.47   197.5 2308.46   214.5 2307.85
   215.7  2307.8225.24512307.877   233.7 2308.33   238.2 2308.03   247.2  2307.8
   251.7 2307.95   256.2 2308.79   260.7 2310.24   269.7 2311.73   280.6 2315.32
   287.7 2317.08   314.7 2321.19   322.2 2321.88   328.2 2322.72   335.8 2323.38
#Mann= 5 ,-1,0
       0     .05       0      70     .07       0   214.5    .045       0
225.2451     .07       0  246.57      .1       0
#XS Ineff= 2 , 0
          144.85 2313.82
Permanent Ineff=
       F       F
Bank Sta=214.5,225.2451
XS Rating Curve= 0 ,0
Exp/Cntr(USF)=0,0
Exp/Cntr=0.3,0.1

Type RM Length L Ch R = 1 ,1230    ,213.3,220,225.9
XS GIS Cut Line= 2
2263191.44972127488128.895098632 2263022.5455954487890.402472904
#Sta/Elev= 30
       0 2320.77    24.2 2319.21    38.9 2317.66    53.6 2317.32    88.7 2314.46
    99.7 2312.97   108.3 2310.93   112.4  2310.6   119.8  2310.9   122.7  2310.8
   130.2 2309.39   144.1 2306.25     151 2305.68   156.5 2306.25     160 2306.86
   171.2 2307.38   176.1 2307.96   178.7 2308.01   195.7 2307.28   213.3 2306.93
   220.2  2307.5   225.1 2308.18   231.7 2308.18   240.3 2308.81     246 2309.58
   257.5 2311.92   266.1 2312.95   274.1 2314.43   280.5 2316.15   292.2 2319.65
#Mann= 6 ,-1,0
       0     .05       0     100     .07       0   144.1    .045       0
   156.5     .07       0     160     .05       0     270      .1       0
Bank Sta=144.1,156.5
XS Rating Curve= 0 ,0
Exp/Cntr(USF)=0,0
Exp/Cntr=0.3,0.1

Type RM Length L Ch R = 1 ,1010    ,97.6,92.8,88.9
XS GIS Cut Line= 4
2263301.57521133488052.5504337392263246.85027455487938.371244651
2263246.85027455487855.9460312262263188.07163875487793.789312906
#Sta/Elev= 30
       0 2319.99    21.5 2319.07    57.6  2316.7    69.5 2315.48    79.1 2313.47
      88 2312.01   119.1 2307.78   127.8 2307.17   143.8 2305.52   155.8 2305.34
   159.8 2304.78   171.8 2303.74   175.8 2303.75   180.82302.969   183.8 2302.35
   187.8 2302.18   191.8 2303.05   199.8  2305.4   207.8 2307.23   212.8 2307.51
   218.6 2307.12   224.6 2307.42   229.4 2308.23   234.9 2310.06   246.8 2312.58
   253.7 2313.77     261 2314.71   272.3 2317.02   280.8 2317.29   294.6 2318.71
#Mann= 4 ,-1,0
       0     .05       0      60      .1       0   180.8    .045       0
   191.8      .1       0
Bank Sta=180.8,191.8
XS Rating Curve= 0 ,0
Exp/Cntr(USF)=0,0
Exp/Cntr=0.3,0.1

Type RM Length L Ch R = 1 ,917     ,106.5,98.8,91.4
XS GIS Cut Line= 3
2263399.46461874 488000.599965942263307.66343332 487802.94639324
 2263243.9646516487780.464470279
#Sta/Elev= 30
       0  2320.1    12.6 2319.06    39.1 2318.18    43.5 2317.67    68.3 2313.47
    78.7 2312.64    83.2 2311.99    87.6 2310.51    96.4 2308.23   100.8 2307.66
   110.5 2307.45   118.4 2306.59   127.3 2303.71  139.542301.251   143.6 2300.91
   149.3 2301.27   162.5 2301.67     167 2302.61   171.4 2303.21   178.7 2303.69
   185.7 2304.48   197.9 2306.71   203.8 2307.53   218.9 2307.88   230.1 2309.54
   242.8 2309.37   247.1 2309.56     264 2311.82     281 2313.68   285.5 2313.97
#Mann= 4 ,-1,0
       0     .05       0     110      .1       0  139.54    .045       0
   149.3      .1       0
Bank Sta=139.54,149.3
XS Rating Curve= 0 ,0
Exp/Cntr(USF)=0,0
Exp/Cntr=0.3,0.1

Type RM Length L Ch R = 1 ,818     ,99.6,93.2,86.7
XS GIS Cut Line= 3
2263500.64973534487840.5749450322263371.83932769487787.519253945
2263293.46781329487746.496157662
#Sta/Elev= 30
       0 2320.11    12.2 2319.87    26.5 2320.18    48.1 2319.66    56.8 2319.87
    65.4 2318.85    70.4 2317.63    82.7 2312.58    85.7 2311.03    88.8 2309.13
     100 2300.93  103.18 2299.66   104.3  2299.3   121.6  2298.9   124.1 2299.54
   130.3 2301.57   134.6 2302.62   143.4 2302.93   155.6 2304.34   170.5 2305.25
   187.5 2305.31   193.1 2305.58   200.1  2306.4   206.7 2307.85   211.9 2308.31
   214.9 2308.41   220.2 2307.74     222 2307.88   223.8 2308.22   227.8 2309.67
#Mann= 3 ,-1,0
       0      .1       0  103.18    .045       0   124.1      .1       0
Bank Sta=103.18,124.1
XS Rating Curve= 0 ,0
Exp/Cntr(USF)=0,0
Exp/Cntr=0.3,0.1

Type RM Length L Ch R = 1 ,725     ,125.8,132.4,140.2
XS GIS Cut Line= 3
2263548.79577408487682.5535925712263370.00940561487716.537778312
2263298.10083868487694.374178916
#Sta/Elev= 30
       0 2321.73      21 2321.25    53.6    2321    57.6 2320.62    65.8 2320.34
    73.9 2320.77    98.4 2318.25   106.5 2316.21   110.6 2314.81   119.1 2310.45
   126.9  2305.6   130.9 2303.43   143.1 2300.51   147.2 2299.31   151.3 2298.05
   155.4 2298.69   156.7  2299.4   159.4 2300.73   163.6 2301.62   171.6 2301.94
   179.8 2302.71   188.1 2302.79   200.7 2303.83     209 2304.22   221.6 2306.08
   229.9 2305.71   234.1 2305.87   237.3 2306.71   242.5 2308.87   257.2 2311.12
#Mann= 4 ,-1,0
       0     .06       0      21      .1       0   147.2    .045       0
   156.7      .1       0
Bank Sta=147.2,156.7
XS Rating Curve= 0 ,0
Exp/Cntr(USF)=0,0
Exp/Cntr=0.3,0.1

Type RM Length L Ch R = 1 ,593     ,127.7,129,130
XS GIS Cut Line= 4
2263523.18450366487655.9572732942263452.26098559487595.376768277
2263375.42717435 487563.855204692263335.04017101487528.393445655
#Sta/Elev= 30
       0 2322.04    14.5 2322.08    26.8  2321.6    30.3  2321.1    35.3 2319.61
    43.8 2317.54    49.5 2315.65    59.7 2311.52    67.1  2308.9    77.6 2304.45
    83.5 2302.44    93.3 2300.03    98.1 2298.34     102 2297.26   110.7 2296.28
   119.3 2294.76     128 2294.24   137.9 2294.67   140.9  2294.9   145.3 2295.79
   153.9 2299.05   158.2 2299.99   166.9 2302.44   175.5 2303.94   180.7 2305.47
   192.5 2309.73   196.6 2310.79     206  2312.9   212.6 2314.05   230.1 2316.11
#Mann= 3 ,-1,0
       0      .1       0   119.3    .045       0   137.9      .1       0
Bank Sta=119.3,137.9
XS Rating Curve= 0 ,0
Exp/Cntr(USF)=0,0
Exp/Cntr=0.3,0.1

Type RM Length L Ch R = 1 ,464     ,88.4,90,90.8
XS GIS Cut Line= 3
 2263569.7395353487568.1420560212263499.54333097487481.603624706
2263391.97064442487421.690449691
#Sta/Elev= 30
       0 2320.69     6.1 2319.38    15.2 2316.18    27.9 2312.46    48.7 2304.36
    65.6  2298.6    77.2 2296.71    91.4 2295.25    97.7 2294.99   117.2 2295.39
     129 2293.27  140.73 2291.98   145.2 2291.67   149.5 2291.82   155.4 2292.11
   158.3  2292.9   161.1 2294.59   164.2 2297.45   167.2 2299.68   170.2 2301.53
     173 2302.46   174.8 2302.85     184 2302.86   186.3 2303.32   197.7 2308.05
   202.4 2309.76   205.4 2310.45     216 2311.84     226 2312.59   234.6 2314.07
#Mann= 3 ,-1,0
       0      .1       0  140.73    .045       0   149.5      .1       0
#XS Ineff= 2 , 0
          124.17 2301.18
Permanent Ineff=
       F       F
Bank Sta=140.73,149.5
XS Rating Curve= 0 ,0
Exp/Cntr(USF)=0,0
Exp/Cntr=0.3,0.1

Type RM Length L Ch R = 1 ,374     ,70.3,69.6,69.1
XS GIS Cut Line= 2
 2263630.6511325487475.771460065 2263448.7907121487346.910362179
#Sta/Elev= 30
       0 2313.79    11.4 2309.43    32.3 2300.86    40.9 2298.01    46.7 2296.84
      61 2295.37    66.8 2294.44    76.6 2293.68    86.4 2293.39    98.3 2294.03
   109.8 2293.72   110.9 2293.58   115.8 2291.96   122.1 2290.89   124.1  2290.9
   135.4 2291.83   140.3 2291.87   145.2 2291.59   150.1 2290.79     155 2290.16
   158.6 2290.38   161.4 2290.94   169.7 2293.37   174.6 2297.12   178.7 2298.71
   184.6 2299.76   187.3 2300.52   198.7 2304.59     216 2308.64   222.9 2310.58
#Mann= 3 ,-1,0
       0      .1       0   150.1    .045       0   161.4      .1       0
#XS Ineff= 2 , 0
           109.1 2299.44
Permanent Ineff=
       F       F
Bank Sta=150.1,161.4
XS Rating Curve= 0 ,0
Exp/Cntr(USF)=0,0
Exp/Cntr=0.3,0.1

Type RM Length L Ch R = 1 ,304     ,91.6,91.4,91.1
XS GIS Cut Line= 3
2263644.66027109 487441.14119638 2263552.2434451487334.338819826
2263473.37101102487284.529498057
#Sta/Elev= 30
       0 2311.11    17.3 2304.71    25.2 2302.17    31.3 2299.97    37.4  2298.1
    43.5 2296.99      68  2294.5    82.6 2291.77    89.9 2290.85    95.2 2290.76
   100.5 2291.06   110.9 2292.85   116.9 2293.28     123 2292.94   141.3 2290.72
   150.6  2289.2  154.67 2288.08   160.2 2287.46     165 2287.69   165.9 2287.89
   169.7 2289.35   179.2 2295.15   183.9 2297.75   188.5 2298.96   193.4 2299.88
   197.2 2300.88   211.7 2305.19   221.7 2307.83   229.1 2310.31   234.5 2312.41
#Mann= 4 ,-1,0
       0     .06       0      30      .1       0  154.67    .045       0
   165.9      .1       0
#XS Ineff= 2 , 0
          120.77 2298.99
Permanent Ineff=
       F       F
Bank Sta=154.67,165.9
XS Rating Curve= 0 ,0
Exp/Cntr(USF)=0,0
Exp/Cntr=0.3,0.1

Type RM Length L Ch R = 1 ,213     ,50.9,49.7,48.7
XS GIS Cut Line= 2
 2263660.3027541 487293.629656032263524.88067167487212.004118633
#Sta/Elev= 30
       0 2308.25     9.5 2308.23    14.2 2307.69    18.8 2306.35    20.8  2305.1
    23.5 2303.65    29.6 2299.44    32.8 2297.08    37.5 2293.92    42.2 2291.48
    46.9 2289.92      50 2289.15    56.2 2287.23    70.2 2284.7179.041822283.744
    84.2 2283.3489.222252283.859    93.7 2284.24    96.6 2285.55    98.2 2286.54
   105.3 2292.85   108.2 2295.04   112.2  2296.2   126.3 2297.45   131.6 2298.83
   134.5 2300.31   140.3 2304.13   148.1 2308.58   154.3 2312.42   158.1 2314.53
#Mann= 4 ,-1,0
       0     .06       0      40      .1       079.04182    .045       0
89.22225      .1       0
Bank Sta=79.04182,89.22225
XS Rating Curve= 0 ,0
Exp/Cntr(USF)=0,0
Exp/Cntr=0.3,0.1

Type RM Length L Ch R = 1 ,163     ,75.8,81.3,86
XS GIS Cut Line= 2
2263670.40728217487234.2550149552263544.95521815487176.009413806
#Sta/Elev= 30
       0 2304.56     2.5 2304.91     6.9 2305.11    11.3 2304.61    20.6 2302.04
    24.5 2300.11    28.9 2297.23    38.6 2289.84    41.6 2287.82    44.7 2286.29
    53.7 2282.46    55.4 2281.93    59.7 2281.78    64.2  2282.2    65.7 2282.49
    68.8 2283.19    71.8 2284.75    77.8 2288.86    81.8 2292.02    86.3 2294.47
      88 2294.99    92.8 2296.06    95.9 2297.05   107.9 2302.46   112.7 2306.12
   116.9 2309.57   121.5 2312.59     129  2316.8     132 2318.35   138.3 2321.03
#Mann= 4 ,-1,0
       0     .06       0      40      .1       0    53.7    .045       0
    65.7      .1       0
Bank Sta=53.7,65.7
XS Rating Curve= 0 ,0
Exp/Cntr(USF)=0,0
Exp/Cntr=0.3,0.1

Type RM Length L Ch R = 1 ,82      ,36.3,33.7,29.8
XS GIS Cut Line= 3
2263705.35464286487200.2037404372263665.92685131487145.542483974
2263626.94710285487139.717923859
#Sta/Elev= 30
       0 2302.05     3.7 2302.02     8.9 2301.31    11.6 2300.67    13.6 2300.03
    15.7 2299.06    18.5 2297.46    20.2 2296.28    23.5 2293.79    25.9 2291.64
    33.3 2285.52    36.2 2283.47    38.3  2282.3    40.3 2281.59    43.2 2280.84
    48.1 2280.33      53 2280.67    56.7 2281.25      58 2281.61    60.3 2282.72
    62.9 2284.17    72.8 2288.84    81.3 2293.15    85.3 2294.91    89.4 2296.24
    93.4 2296.86    96.9 2296.56   101.5    2296   104.4 2296.03   106.8 2296.24
#Mann= 3 ,-1,0
       0      .1       0    43.2    .045       0      53      .1       0
Bank Sta=43.2,53
XS Rating Curve= 0 ,0
Exp/Cntr(USF)=0,0
Exp/Cntr=0.5,0.3

Type RM Length L Ch R = 1 ,48      ,25.5,25.3,25.4
XS GIS Cut Line= 4
2263730.22105046487195.4747859362263726.41266789487160.327905804
2263658.31011885487108.8029509412263618.88232731487115.075554142
#Sta/Elev= 30
       0 2299.81     2.3 2299.58     6.3 2298.14    10.4 2295.65    14.4 2293.15
    26.4 2286.99    30.5 2285.62    34.5 2285.12    42.1 2284.75    44.9 2284.22
    56.3  2279.8    58.2 2279.42    63.2 2279.33    67.1 2279.36   68.84 2279.78
    78.3 2282.78    84.9 2283.74    87.7 2283.81    93.6 2283.31   110.6 2283.37
   113.4 2283.15   119.2 2283.53   122.9 2283.44     127 2284.46   135.1 2289.12
   139.1 2290.72   143.2 2291.87   147.2  2292.5   155.3  2293.2   160.7 2295.64
#Mann= 4 ,-1,0
       0     .06       0    10.4      .1       0    56.3    .045       0
   68.84      .1       0
#XS Ineff= 2 , 0
              45    2287      76            2286
Permanent Ineff=
       F       F
Bank Sta=56.3,68.84
XS Rating Curve= 0 ,0
Exp/Cntr(USF)=0,0
Exp/Cntr=0.5,0.3

Type RM Length L Ch R = 1 ,23      ,4.3,4.3,4.3
XS GIS Cut Line= 4
2263738.82763361487195.8818276722263736.70747744487136.729470337
2263686.24776043487097.7185966832263612.67834109 487103.44301836
#Sta/Elev= 30
       0 2299.13     2.7 2298.96     6.7  2297.6    18.7 2289.97    26.7 2285.97
    30.7 2285.45    38.7  2286.9    50.7 2287.11    54.7 2285.99    59.2 2283.43
      70 2278.93    70.7 2278.75      75 2278.16    80.1  2278.2    85.1 2278.72
    87.8  2279.8    90.2 2280.01   100.3  2279.6   110.4 2281.14   115.5 2280.59
     123 2280.58   129.1 2283.53   133.1  2284.6   145.1  2284.7   157.1 2283.79
   161.2  2284.2   176.5 2289.53   189.2 2291.45   193.3 2293.04196.7633 2295.24
#Mann= 4 ,-1,0
       0     .06       0      70      .1       0    70.7    .045       0
    85.1      .1       0
#XS Ineff= 2 , 0
              68    2287      96            2286
Permanent Ineff=
       F       F
Bank Sta=70.7,85.1
XS Rating Curve= 0 ,0
Exp/Cntr(USF)=0,0
Exp/Cntr=0.5,0.3
